--- LAURELCK_T1.prj (project) ---

Proj Title=LAURELCK_T1
Current Plan=p01
Default Exp/Contr=0,0
English Units
Geom File=g01
Flow File=f01
Plan File=p01
BEGIN DESCRIPTION:
Stream Name: Laurel Creek Tributary 1
Flood Zone: Approximate
Summers County, West Virginia
HEC-RAS Version: 5.0.7
Hydrology Method:
regression
Model Notes:
coincident peak with LAURELCK_A
END DESCRIPTION:
DSS Export Rating Curves= 0
DSS Export Rating Curve Sorted= 0
DSS Export Volume Flow Curves= 0
DXF OffsetX= 0
DXF OffsetY= 0
DXF ScaleX= 0
DXF ScaleY= 0

--- LAURELCK_T1.p01 (plan) ---

Plan Title=Floodplain
Program Version=5.07
Short Identifier=Floodplain
Geom File=g01
Flow File=f01
Subcritical Flow
K Sum by GR= 0
Std Step Tol= 0.01
Critical Tol= 0.01
Num of Std Step Trials= 20
Max Error Tol= 0.3
Flow Tol Ratio= 0.001
Split Flow NTrial= 30
Split Flow Tol= 0.02
Split Flow Ratio= 0.02
Log Output Level= 0
Friction Slope Method= 1
Unsteady Friction Slope Method= 2
Unsteady Bridges Friction Slope Method= 1
Parabolic Critical Depth
Global Vel Dist= 0 , 0 , 0
Global Log Level= 0
CheckData=True
Encroach Param=-1 ,0,0, 0
Mapping Interval=1HOUR
Computation Time Step Use Courant=        0
Computation Time Step Use Time Series=    0
Computation Time Step Count To Double=0
Computation Time Step Max Doubling=0
Computation Time Step Max Halving=0
Computation Time Step Residence Courant=0
Run HTab= 0
Run UNet= 0
Run Sediment= 0
Run PostProcess= 0
Run WQNet= 0
Run RASMapper= 0
UNET Theta= 0
UNET Theta Warmup= 0
UNET ZTol= 0
UNET ZSATol= 0
UNET MxIter= 0
UNET Max Iter WO Improvement= 0
UNET MaxInSteps= 0
UNET DtIC= 0
UNET DtMin= 0
UNET MaxCRTS= 0
UNET WFStab= 0
UNET SFStab= 0
UNET WFX= 1
UNET SFX= 1
UNET 1D Methodology=Finite Difference
UNET DSS MLevel= 1
UNET Pardiso=0
UNET DZMax Abort= 0
UNET Use Existing IB Tables= 0
UNET Froude Reduction=False
UNET Froude Limit= 0
UNET Froude Power= 0
UNET D1 Cores= 0
UNET D2 Coriolis=0
UNET D2 Cores= 0
UNET D2 Theta= 1
UNET D2 Theta Warmup= 1
UNET D2 Z Tol= 0.01
UNET D2 Volume Tol= 0.01
UNET D2 Max Iterations= 20
UNET D2 Equation= 0
UNET D2 RampUpFraction=0.1
UNET D2 TimeSlices= 1
UNET D2 BCVolumeCheck=0
UNET D1D2 MaxIter= 0
UNET D1D2 ZTol=0.01
UNET D1D2 QTol=0.1
UNET D1D2 MinQTol=1
Write IC File= 0
Write IC File at Fixed DateTime=0
Write IC File at Sim End=0
Echo Input=False
Echo Parameters=False
Echo Output=False
Write Detailed= 0
HDF Write Warmup=0
HDF Write Time Slices=0
HDF Flush=0
HDF Face Node Velocities=0
HDF Compression= 1
HDF Chunk Size= 1
HDF Spatial Parts= 1
HDF Use Max Rows=0
HDF Fixed Rows= 1
Calibration Method= 0
Calibration Iterations= 20
Calibration Max Change=0.05
Calibration Tolerance=0.2
Calibration Maximum=1.5
Calibration Minimum=0.5
Calibration Optimization Method= 1
WQ AD Non Conservative
WQ ULTIMATE=-1
WQ Max Comp Step=1HOUR
WQ Output Interval=15MIN
WQ Output Selected Increments= 0
WQ Output face flow=0
WQ Output face velocity=0
WQ Output face area=0
WQ Output face dispersion=0
WQ Output cell volume=0
WQ Output cell surface area=0
WQ Output cell continuity=0
WQ Output cumulative cell continuity=0
WQ Output face conc=0
WQ Output face dconc_dx=0
WQ Output face courant=0
WQ Output face peclet=0
WQ Output face adv mass=0
WQ Output face disp mass=0
WQ Output cell mass=0
WQ Output cell source sink temp=0
WQ Output nsm pathways=0
WQ Output nsm derived pathways=0
WQ Output MaxMinRange=-1
WQ Daily Max Min Mean=-1
WQ Daily Range=0
WQ Daily Time=0
WQ Create Restart=0
WQ Fixed Restart=0
WQ System Summary=0
WQ Write To DSS=0
WQ Use Fixed Temperature=0
Sorting and Armoring Iterations= 10
XS Update Threshold= 0.02
Bed Roughness Predictor= 0
Hydraulics Update Threshold= 0.02
Energy Slope Method= 1
Volume Change Method= 1
Sediment Retention Method= 0
XS Weighting Method= 0
Number of US Weighted Cross Sections= 1
Number of DS Weighted Cross Sections= 1
Upstream XS Weight=0
Main XS Weight=1
Downstream XS Weight=0
Number of DS XS's Weighted with US Boundary= 1
Upstream Boundary Weight= 1
Weight of XSs Associated with US Boundary= 0
Number of US XS's Weighted with DS Boundary= 1
Downstream Boundary Weight= 0.5
Weight of XSs Associated with DS Boundary= 0.5
Percentile Method= 0
Sediment Output Level= 3
Mass or Volume Output= 0
Output Increment Type= 1
Profile and TS Output Increment= 1
XS Output Flag= 0
XS Output Increment= 10
Write Gradation File= 0
Read Gradation Hotstart= 0
Write HDF5 File= 1
Write Binary Output= 1
Write DSS Sediment File= 0
SV Curve= 0
Specific Gage Flag= 0

--- LAURELCK_T1.f01 (steady flow) ---

Flow Title=Flows
Program Version=5.07
Number of Profiles= 6
Profile Names=01pct,10pct,04pct,02pct,0_2pct,01plus
River Rch & RM=LAURELCK_T1,Main            ,9387
     532     280     373     450     744     787
River Rch & RM=LAURELCK_T1,Main            ,8584
     592     313     416     501     826     876
River Rch & RM=LAURELCK_T1,Main            ,6701
     819     439     579     695    1136    1211
River Rch & RM=LAURELCK_T1,Main            ,2525
     966     521     686     822    1336    1429
River Rch & RM=LAURELCK_T1,Main            ,0
    1881    1041    1353    1609    2569    2781
Boundary for River Rch & Prof#=LAURELCK_T1,Main            , 1
Up Type= 0
Dn Type= 1
Dn Known WS=1785.8
Boundary for River Rch & Prof#=LAURELCK_T1,Main            , 2
Up Type= 0
Dn Type= 1
Dn Known WS=1784.2
Boundary for River Rch & Prof#=LAURELCK_T1,Main            , 3
Up Type= 0
Dn Type= 1
Dn Known WS=1784.7
Boundary for River Rch & Prof#=LAURELCK_T1,Main            , 4
Up Type= 0
Dn Type= 1
Dn Known WS=1785.4
Boundary for River Rch & Prof#=LAURELCK_T1,Main            , 5
Up Type= 0
Dn Type= 1
Dn Known WS=1786.8
Boundary for River Rch & Prof#=LAURELCK_T1,Main            , 6
Up Type= 0
Dn Type= 1
Dn Known WS=1787
DSS Import GetInterval= 0
DSS Import GetPeak= 0
DSS Import FillOption= 0

--- LAURELCK_T1.g01 (geometry) ---

Geom Title=Geometry
Program Version=5.07

River Reach=LAURELCK_T1     ,Main
Reach XY= 30
2023948.83946665267106.577267186     2023858.809267157.671999915
2023830.00099999 267303.807999912023588.90099999267404.762999913
2023172.51499999267808.4359999182022903.36199999267829.536999916
2022788.77299999268089.8519999152022582.78599999268139.855999905
2022523.80599999268502.679999907     2022287.695268774.901999913
 2022225.8176624269030.4019794562022277.97199999269289.228999923
2022157.23638778 269454.070548382022078.76823638270064.951079566
2022327.94489855270231.4286554882022385.53799999270649.925999912
     2022570.595270746.6299999082022735.01399999271010.784999913
     2022733.484271263.4959999132022923.53935805271611.536729669
2022928.44208098271782.9452837922022733.70099999272004.936999917
2022745.95199999272312.038999912     2022626.931 272739.31199991
2022117.38199999 272899.03399991     2022084.396273146.429999916
2021900.36799999273143.825999917     2021743.941273354.884999913
2021613.90999999273874.7289999062021362.85339825274038.742884472

Type RM Length L Ch R = 1 ,9387    ,172.4,163.3,142.3
XS GIS Cut Line= 2
2023890.59125972266998.2911282372024025.02324199267287.880100525
#Sta/Elev= 30
       0 2225.69    10.2  2218.3    31.9 2200.29    40.5 2194.33    53.6 2187.48
    75.4 2178.16    89.8  2169.2   102.8 2160.34   104.3 2159.66   111.5 2159.06
   122.4 2157.78     131 2158.71   133.2 2159.61   136.8 2162.76   138.4 2163.53
   140.5 2164.26   151.3 2165.95   165.8 2164.71   180.7 2165.92   232.3 2164.42
     249 2164.54   259.8 2165.29   267.1 2166.87   274.3 2170.18   279.2 2172.89
   289.1  2179.6   292.4 2181.17     296  2182.2   306.8 2184.01   319.3 2184.39
#Mann= 3 ,-1 , 0
       0      .1       0   111.5    .045       0     131      .1       0
Bank Sta=111.5,131
XS Rating Curve= 0 ,0
Exp/Cntr=0.3,0.1

Type RM Length L Ch R = 1 ,9223    ,216,238.8,258.2
XS GIS Cut Line= 4
2023733.47072058267133.0651409612023763.63481727267204.267916205
2023954.96685184 267233.239328382023976.84265427267301.721009796
#Sta/Elev= 30
       0 2202.42    20.5 2196.14    45.4 2183.72    62.2 2172.67    73.9 2163.42
    77.3  2161.2    86.9 2157.49    94.5 2155.88   116.8 2155.87   130.1 2156.69
   133.4 2155.42     140 2148.29   143.4 2145.67   146.7 2144.74     150 2144.51
   156.6 2144.69   163.6 2145.63   169.9 2146.25   179.8 2146.07   189.8 2149.81
   209.7  2151.6     227 2157.85   270.8 2161.18   292.3 2162.02   295.7 2162.84
   301.6 2165.52   312.9 2172.49   319.8 2175.95     333 2179.21   342.7 2179.39
#Mann= 3 ,-1 , 0
       0      .1       0   143.4    .045       0   163.6      .1       0
Bank Sta=143.4,163.6
XS Rating Curve= 0 ,0
Exp/Cntr(USF)=0,0
Exp/Cntr=0.3,0.1

Type RM Length L Ch R = 1 ,8984    ,242.5,233.3,223.1
XS GIS Cut Line= 2
2023673.18794823267217.1527413312023722.29258405267467.606487343
#Sta/Elev= 30
       0 2191.28    11.1 2188.13    20.5 2183.32    37.2 2172.02    47.2 2164.16
    70.6 2149.65    77.1 2146.76    87.3 2143.39   104.1 2140.27   110.7 2136.81
   117.4 2135.28   124.1 2135.16   127.5 2133.91   134.1 2128.03   135.8 2127.57
   135.8 2127.56   140.8 2126.97   164.2 2127.63   167.6  2128.9   170.9 2131.06
   180.9 2139.99   184.3 2142.63   187.6  2144.3     191 2144.73     211 2144.39
   221.1 2142.66   224.4 2143.72     228 2146.47   231.1 2147.76   255.2 2149.32
#Mann= 3 ,-1 , 0
       0      .1       0   135.8    .045       0   164.2      .1       0
Bank Sta=135.8,164.2
XS Rating Curve= 0 ,0
Exp/Cntr=0.3,0.1

Type RM Length L Ch R = 1 ,8751    ,165.4,166.7,167.9
XS GIS Cut Line= 2
2023422.76149508267374.1081550962023574.40748063267555.671416419
#Sta/Elev= 30
       0 2162.74    26.9 2158.37    39.8 2155.43    50.1 2154.15    65.3 2150.98
    73.9 2149.55    78.2 2148.36   102.7 2140.02     119 2133.13   120.9 2132.22
     132 2125.38   142.2 2118.23   146.5 2116.53   149.2 2115.92   153.9 2115.35
   165.5 2115.47   167.9 2115.61   170.2 2116.19   172.2 2116.74   178.1 2120.21
   180.7 2121.36     185 2121.89   198.5 2122.26   206.4 2123.16   210.7 2124.11
   214.5 2125.79   219.1 2128.44   221.4 2129.13   224.1 2129.57   236.6  2129.7
#Mann= 3 ,-1 , 0
       0      .1       0   149.2    .045       0   170.2      .1       0
Bank Sta=149.2,170.2
XS Rating Curve= 0 ,0
Exp/Cntr=0.3,0.1

Type RM Length L Ch R = 1 ,8584    ,127.5,122.7,118.6
XS GIS Cut Line= 2
2023306.33152271267465.6118804442023440.25651567267661.668438116
#Sta/Elev= 30
       0  2143.2     5.5 2143.37    29.9 2140.48    67.7 2137.48    77.2 2135.24
      85 2134.29   110.2 2133.93   119.6  2132.9     122 2132.07   124.7 2130.52
   128.7 2126.49   136.6 2117.28   143.2 2111.12     147 2108.63   150.3 2107.37
   157.4 2106.15   162.1 2106.44   168.4 2107.83   172.4 2108.27   176.4 2109.41
   183.4 2113.18   192.3 2119.05   196.2 2120.63   199.9 2121.16   208.2  2121.3
   216.8 2120.52   220.1 2121.13   224.1 2123.08   225.8 2123.48   237.4 2124.94
#Mann= 3 ,-1 , 0
       0      .1       0   150.3    .045       0   168.4      .1       0
Bank Sta=150.3,168.4
XS Rating Curve= 0 ,0
Exp/Cntr=0.3,0.1

Type RM Length L Ch R = 1 ,8462    ,78.7,76,69.9
XS GIS Cut Line= 2
2023146.77740591 267541.82398907  2023384.775203267734.281442292
#Sta/Elev= 30
       0 2132.93    18.8 2126.79    29.2 2124.04    37.4  2120.8    42.2 2117.64
    50.3 2110.73    53.8 2108.89    92.5 2111.14   105.2  2110.6   117.8  2107.4
   130.4 2106.83   157.4 2109.51   165.8 2107.46   178.2 2102.29   183.5 2101.08
   188.7 2100.88   197.9 2102.35   206.4 2103.97   209.6 2105.29   214.8 2108.63
     220 2110.58   235.6 2111.66   246.1 2110.73   248.6  2112.6   252.8 2117.35
     257 2120.95   261.7  2122.5   278.1 2125.92   289.4 2129.68   306.1 2132.87
#Mann= 3 ,-1 , 0
       0      .1       0   178.2    .045       0   197.9      .1       0
Bank Sta=178.2,197.9
XS Rating Curve= 0 ,0
Exp/Cntr(USF)=0,0
Exp/Cntr=0.5,0.3

Type RM Length L Ch R = 1 ,8386    ,40.2,39.7,40.6
XS GIS Cut Line= 3
2023155.11446658267603.599444225 2023182.0954653267689.839659255
2023360.06844035267759.022763248
#Sta/Elev= 30
       0 2104.12       8 2104.85    32.1 2103.62      63 2105.26      70  2104.7
    80.2 2103.25    90.4 2101.32   106.1 2100.18   122.6 2099.76   136.6 2100.86
   140.2 2100.75   143.7 2100.08   147.2 2099.23   154.2 2098.65   161.3 2098.98
   166.9 2100.08   174.5 2102.25     177 2102.55   199.5 2103.66     207 2103.02
   208.5 2103.32   210.6 2104.35   217.6 2110.51   220.1 2112.32   227.7 2116.45
   235.2 2119.08   242.2 2122.75   245.8 2124.15   266.9 2129.56   281.3 2135.37
#Mann= 3 ,-1 , 0
       0      .1       0   143.7    .045       0   166.9      .1       0
#XS Ineff= 3 ,-1
  135.49     140  2097.4      77  135.49 2102.72     184   281.3  2101.2
Permanent Ineff=
       F       F       F
Bank Sta=143.7,166.9
XS Rating Curve= 0 ,0
Exp/Cntr(USF)=0,0
Exp/Cntr=0.5,0.3

Type RM Length L Ch R = 1 ,8346    ,96.5,106.3,116.3
XS GIS Cut Line= 3
2023139.85796921267605.1558053132023171.46778345267726.479127515
2023340.04487035267790.485170016
#Sta/Elev= 30
       0 2105.55     2.9 2103.79     6.3 2103.01    16.5 2103.55    50.4 2101.27
    77.5 2101.52    84.3 2100.51    91.1 2100.12     108 2096.33   136.2 2096.87
   154.8  2098.9   158.3 2098.78   165.3  2096.6   171.8    2096     182 2096.57
   192.2 2097.74   197.3 2099.43   203.9 2102.28   214.5 2103.55     218 2104.63
   225.9 2107.54     239 2113.86   248.1 2117.41   256.6 2120.32   263.6 2121.95
   274.1 2126.52   281.4 2128.95   291.7 2134.27   295.2  2135.7   305.7 2138.12
#Mann= 3 ,-1 , 0
       0      .1       0   165.3    .045       0     182      .1       0
#XS Ineff= 2 , 0
          153.73 2100.26
Permanent Ineff=
       F       F
Bank Sta=165.3,182
XS Rating Curve= 0 ,0
Exp/Cntr(USF)=0,0
Exp/Cntr=0.5,0.3

Type RM Length L Ch R = 1 ,8240    ,204.1,206.9,203.3
XS GIS Cut Line= 3
2022980.81129127267652.4291150462023110.17608145267750.820543733
2023200.24905926267911.326515847
#Sta/Elev= 30
       0 2107.18    16.3 2103.68    20.9 2103.24    47.4 2104.44    77.1 2103.61
   105.1 2104.23   109.9 2102.83   126.3 2094.12     134 2092.05   154.2 2091.92
   180.7 2093.82   201.9 2094.06   209.9 2094.88   214.4 2094.28     224  2089.6
   230.3 2087.64   240.9 2086.72   251.42087.653   254.6 2089.84   262.1 2102.03
     265 2105.78   269.6 2110.58   289.1 2133.41   293.9 2138.23     311 2150.61
   314.7 2151.79   322.3 2151.86   325.3  2152.8   333.6 2159.37   346.6 2165.75
#Mann= 3 ,-1 , 0
       0      .1       0   230.3    .045       0   251.4      .1       0
Bank Sta=230.3,251.4
XS Rating Curve= 0 ,0
Exp/Cntr(USF)=0,0
Exp/Cntr=0.3,0.1

Type RM Length L Ch R = 1 ,8033    ,283.8,267.4,242.6
XS GIS Cut Line= 3
2022889.68916562267579.7954735572022898.85039127267694.913924168
2023011.00523462267944.011362127
#Sta/Elev= 30
       0 2139.47    31.6 2126.44    54.6 2120.61    77.6 2116.43    90.8 2113.37
   119.3 2109.78   142.5  2105.7   189.2 2100.31   192.8 2098.99   199.8 2095.19
   203.6 2092.53   207.2 2088.84   210.8 2086.92   222.1 2086.82   225.2 2085.41
   228.8 2082.22   231.2  2080.6   232.4 2079.85     237 2079.15   257.6 2080.63
   279.1 2084.44   291.6 2084.18   297.2  2084.7   318.9 2091.83   333.8 2095.74
   343.7 2099.32   359.1 2106.44   373.5 2114.54   383.5 2121.59   388.7 2123.11
#Mann= 3 ,-1 , 0
       0      .1       0   231.2    .045       0   257.6      .1       0
Bank Sta=231.2,257.6
XS Rating Curve= 0 ,0
Exp/Cntr=0.3,0.1

Type RM Length L Ch R = 1 ,7765    ,256.3,280.5,299.8
XS GIS Cut Line= 4
2022548.15607145267820.9373277052022684.02166547268011.079937642
2022907.49378314268032.1009460772022987.43853621268112.148663201
#Sta/Elev= 30
       0  2103.4     8.1 2100.65    24.6 2096.72    64.2 2089.04    78.7  2087.1
   153.6 2080.25   189.2 2078.86   203.3 2079.27   218.1 2078.57   226.9 2075.68
   266.5 2077.34   286.3 2072.53   325.8 2072.52   335.7 2069.42   348.9  2070.5
   358.8 2065.99     372  2064.8   391.7 2066.42     395 2068.01   404.9 2077.79
   411.5 2082.62   434.6 2092.09   458.2 2104.65   480.4 2120.54   487.3 2127.03
   499.2 2134.87   517.2 2145.11   554.3 2167.63   563.5 2174.11   571.3 2175.59
#Mann= 3 ,-1 , 0
       0      .1       0   358.8    .045       0   391.7      .1       0
Bank Sta=358.8,391.7
XS Rating Curve= 0 ,0
Exp/Cntr=0.3,0.1

Type RM Length L Ch R = 1 ,7485    ,211.4,195.2,182.3
XS GIS Cut Line= 2
  2022463.163902267900.5498632572022683.02899846268292.443298792
#Sta/Elev= 30
       0 2101.34    24.3 2094.19    43.6 2091.85      52 2087.87    65.3  2084.7
    77.4 2083.09      87 2080.57   108.7 2078.09   129.3 2072.97   161.1 2071.78
   168.6 2070.52   179.9 2071.14   195.4 2070.46   202.5 2069.53   213.8 2065.33
   221.3 2063.63   240.1  2062.5   243.9 2061.38   255.1  2052.9   258.1  2051.8
   267.7 2050.84   276.8 2051.93   285.2 2053.63   303.9 2054.45   345.4 2065.54
   364.1 2068.27   377.4 2071.94   393.1  2077.7   401.9 2081.75   449.4 2107.45
#Mann= 3 ,-1 , 0
       0      .1       0   258.1    .045       0   276.8      .1       0
#XS Ineff= 2 , 0
                             295            2056
Permanent Ineff=
       F       F
Bank Sta=258.1,276.8
XS Rating Curve= 0 ,0
Exp/Cntr(USF)=0,0
Exp/Cntr=0.3,0.1

Type RM Length L Ch R = 1 ,7290    ,197.8,206.1,214.5
XS GIS Cut Line= 2
 2022220.4668548268271.8449106522022673.07617472268322.441480968
#Sta/Elev= 30
       0 2072.77    20.6 2069.99    66.9 2067.44    85.8 2065.25    99.9 2064.18
   119.7 2063.97   136.2 2062.04   179.1 2061.84   208.8 2060.28   231.3  2058.6
   235.2 2057.93   238.5 2056.81   261.6 2046.17   264.9 2045.04   278.1 2042.86
   281.4 2042.39   297.9 2041.83   303.3 2042.94   310.7 2045.54   314.4  2047.4
   317.8 2048.48   324.4 2049.25     331 2051.87   350.1 2062.83   360.7 2068.33
   381.3 2076.22   406.9 2085.34   433.2  2098.2   449.8 2105.32   455.4  2108.4
#Mann= 5 ,-1 , 0
       0      .1       0      50     .04       0     220      .1       0
   278.1    .045       0   303.3      .1       0
Bank Sta=278.1,303.3
XS Rating Curve= 0 ,0
Exp/Cntr(USF)=0,0
Exp/Cntr=0.3,0.1

Type RM Length L Ch R = 1 ,7084    ,209.2,214.4,218
XS GIS Cut Line= 2
 2022369.3593544268405.3882686192022652.86011471 268593.72330002
#Sta/Elev= 30
       0 2051.94    54.6 2049.43    58.6 2048.75    66.4 2044.72    82.4 2039.79
      98 2038.43   117.6 2038.48   121.6  2037.6   130.1 2034.23     161 2033.77
   168.9 2031.62   174.7  2030.3   188.5 2029.46   192.5 2030.48   193.6 2031.42
   196.4 2033.59   200.4 2038.93   208.2  2053.2   213.1 2060.71     224    2073
   235.8  2084.7   242.8 2090.18   252.8 2096.84   276.5 2107.92   283.1  2114.3
   294.9  2131.6     308  2139.2   314.6 2143.93   321.4 2149.82   340.4 2162.94
#Mann= 3 , 0 , 0
       0      .1       0   168.9    .045       0   193.6      .1       0
Bank Sta=168.9,193.6
XS Rating Curve= 0 ,0
Exp/Cntr(USF)=0,0
Exp/Cntr=0.3,0.1

Type RM Length L Ch R = 1 ,6869    ,177.8,168.4,162.5
XS GIS Cut Line= 2
2022221.14080219268472.9770079592022505.94656773268810.696449754
#Sta/Elev= 30
       0 2051.22     5.3  2049.2    10.1 2048.23    28.9 2045.74      53 2041.72
    61.3 2040.94    76.6 2040.11   117.4 2039.82   181.7 2036.07   203.8 2033.42
   216.1  2031.1   236.1 2024.54   252.4 2017.94     257 2016.95     264 2016.68
   271.9 2017.66   280.1 2020.55   284.7 2021.21   300.5 2021.26   310.7 2022.46
   323.4 2026.98     332 2031.76   353.4 2046.75   366.5 2054.45   374.9 2060.38
   397.2 2079.99   402.3 2085.27   409.2 2093.65   417.5 2102.12   441.8  2121.5
#Mann= 4 ,-1 , 0
       0     .04       0      30      .1       0   252.4    .045       0
   271.9      .1       0
Bank Sta=252.4,271.9
XS Rating Curve= 0 ,0
Exp/Cntr=0.3,0.1

Type RM Length L Ch R = 1 ,6701    ,230.2,233.1,236
XS GIS Cut Line= 2
2022109.11837265268744.5616101122022451.14198861268847.392239746
#Sta/Elev= 30
       0 2037.75    14.4 2033.01    41.8 2020.93    55.5 2017.65    65.7  2016.3
    74.8 2016.02    79.4 2016.93    93.2  2021.7   103.4  2022.4   113.7 2020.54
   128.4 2015.83   141.1 2013.24     148 2012.91   151.4 2011.94   154.8 2010.18
   168.2 2009.34   182.2 2008.86   184.62009.471   192.5 2011.12   202.8 2011.36
   213.1 2010.43   233.6 2006.97   244.3 2008.17   250.7  2011.1   254.2  2013.5
     261 2020.79   271.3 2030.12   312.4 2059.07   336.2  2076.6   357.1 2093.69
#Mann= 4 ,-1 , 0
       0     .04       0      40      .1       0   168.2    .045       0
   184.6      .1       0
#XS Ineff= 2 , 0
                          202.94          2014.5
Permanent Ineff=
       F       F
Bank Sta=168.2,184.6
XS Rating Curve= 0 ,0
Exp/Cntr(USF)=0,0
Exp/Cntr=0.3,0.1

Type RM Length L Ch R = 1 ,6468    ,224.2,215.8,204.6
XS GIS Cut Line= 3
2022088.74928167268952.9585258212022318.73369219269051.391853526
2022416.24708225269044.952290032
#Sta/Elev= 30
       0 2029.34    19.3  2028.1      30 2025.48    40.7 2020.64    48.6 2017.97
    62.1 2012.36    72.8 2008.31    83.5 2005.28    90.6 2002.36    94.2 2001.45
   108.5 1995.52   126.3 1993.59   133.5 1993.71   143.6 1992.33   151.3 1991.22
   156.1 1991.19   163.6 1991.32   171.1 1992.56   176.3  1993.4   183.5 1996.69
   195.6 1999.15   208.9 2003.02   222.7  2008.3   229.8 2011.78   247.7 2022.39
   264.3 2033.41   297.2 2052.96   323.5 2070.02   335.9 2078.87   347.9 2088.58
#Mann= 4 ,-1 , 0
       0     .04       0      60      .1       0   143.6    .045       0
   171.1      .1       0
#XS Ineff= 2 , 0
             129    1999
Permanent Ineff=
       F       F
Bank Sta=143.6,171.1
XS Rating Curve= 0 ,0
Exp/Cntr(USF)=0,0
Exp/Cntr=0.3,0.1

Type RM Length L Ch R = 1 ,6252    ,283.1,291.1,277.9
XS GIS Cut Line= 2
2022031.46879758269253.1685944112022508.61346529269192.177221739
#Sta/Elev= 30
       0 2006.55    12.8 2006.05    22.7 2002.89    52.5 2000.39    85.5 2000.56
   128.5 1999.74   181.4 2000.85   201.3 1992.66   214.5 1988.58   224.4 1982.63
   227.8 1982.11   255.41982.369   267.4 1983.31   279.5  1991.4   290.6    1996
   300.5 2003.33   320.4 2014.37   335.2 2027.57   352.8 2040.51   361.6 2048.11
   373.2 2055.96   383.2  2064.3   409.7 2083.75   426.2 2096.97   439.4 2106.23
   446.7 2110.58   449.4 2112.87   458.4 2123.44   475.8 2138.43     481 2144.13
#Mann= 4 ,-1 , 0
       0     .04       0      10      .1       0   224.4    .045       0
   255.4      .1       0
Bank Sta=224.4,255.4
XS Rating Curve= 0 ,0
Exp/Cntr=0.3,0.1

Type RM Length L Ch R = 1 ,5961    ,247.9,251.1,248.8
XS GIS Cut Line= 3
2021996.91781469269480.8926600092022345.41188381269460.764104262
2022524.79972402269398.208344599
#Sta/Elev= 30
       0 2017.84    27.6 2005.05    37.4 1997.99    47.3 1989.36    50.6 1988.54
    64.6 1988.61    83.4 1977.68      90 1976.58   109.7 1976.95   132.7 1975.53
   142.6 1973.54   149.2 1970.74     159 1969.25   178.7 1970.46   188.6 1969.58
   193.4 1970.57   199.6  1972.3     228 1975.26   237.9 1977.49   254.3 1976.58
   283.9 1977.13   290.5 1977.95   302.2 1981.17   313.5 1987.73   339.4 2004.86
   349.7 2009.84   394.8 2026.95   431.3 2043.44   475.1 2065.86   539.1 2102.67
#Mann= 4 ,-1 , 0
       0      .1       0      50     .04       0   149.2    .045       0
   193.4      .1       0
Bank Sta=149.2,193.4
XS Rating Curve= 0 ,0
Exp/Cntr(USF)=0,0
Exp/Cntr=0.3,0.1

Type RM Length L Ch R = 1 ,5710    ,237.8,251.8,265.9
XS GIS Cut Line= 3
2021916.26363765269725.6176076172022243.72693727269701.528142318
2022394.86233395269638.452412103
#Sta/Elev= 30
       0 2006.65    55.8 1991.16    65.7 1988.06    72.3 1985.35   101.9 1970.94
   115.5 1966.92   124.9 1962.78   141.4 1963.43   154.5 1962.53   164.4 1960.64
     171 1960.07   184.1 1960.68   210.5 1960.95     217 1960.25   223.51959.011
   230.2  1957.4   233.5 1957.24   243.3  1957.8     2481959.796   255.7 1964.58
   268.1 1971.41   276.2 1975.04   279.5 1976.02   302.6 1978.19   346.4 1983.22
   410.7  1991.8   428.5 1995.13   449.4 2000.39   464.5 2003.52   492.1 2010.09
#Mann= 4 ,-1 , 0
       0      .1       0     130     .04       0   223.5    .045       0
     248      .1       0
#XS Ineff= 2 , 0
             208    1964
Permanent Ineff=
       F       F
Bank Sta=223.5,248
XS Rating Curve= 0 ,0
Exp/Cntr(USF)=0,0
Exp/Cntr=0.5,0.3

Type RM Length L Ch R = 1 ,5458    ,42.2,44.6,47.2
XS GIS Cut Line= 4
2021920.17181055269892.8282430562022058.82391923269902.396848641
2022117.22235927269972.3889664732022293.08223129269901.675677763
#Sta/Elev= 30
       0 1993.82    22.3 1985.99      42 1979.85    68.3 1967.59    81.5  1962.1
    88.1 1957.69    91.4 1955.96   101.2  1952.3     121 1947.16   146.8 1946.78
   158.9 1947.17   167.3 1946.51   172.4 1944.95   177.5 1942.44   180.3 1941.63
   182.6 1940.97   187.7 1940.55   193.1 1941.49   205.9 1945.43   220.9 1947.15
   230.1 1947.63   236.3 1952.09   239.8  1953.7   243.3 1954.46   284.1 1955.25
   296.3 1956.63   345.8 1960.26   388.3 1961.99     406 1966.18   419.7 1970.74
#Mann= 5 ,-1 , 0
       0      .1       0     130     .04       0   180.3    .045       0
   193.1     .04       0  260.14      .1       0
#XS Ineff= 3 ,-1
       0   170.3  1946.5     200     205  1944.4     205  419.68  1946.5
Permanent Ineff=
       F       F       F
Bank Sta=180.3,193.1
XS Rating Curve= 0 ,0
Exp/Cntr(USF)=0,0
Exp/Cntr=0.5,0.3

Type RM Length L Ch R = 1 ,5414    ,273.8,251.9,222.8
XS GIS Cut Line= 4
2021923.51197899269932.7093293782022034.79935757269928.076094393
2022130.22602875270034.9488816232022315.39050838269961.398958355
#Sta/Elev= 30
       0 2000.11    28.8 1991.19    48.5 1982.67    62.3  1974.4    84.6 1958.75
    97.7 1952.52   104.3  1950.7   115.5 1949.17   130.3 1949.57   135.2 1949.05
   145.1 1946.08   150.1  1946.2   159.9 1945.09   169.7 1941.11   174.6 1940.34
   184.5 1939.24   189.4 1939.37   196.6 1940.76   204.2 1942.39   253.5 1940.51
     275  1942.8   296.3 1942.89     309 1945.25   334.2 1954.19   364.6 1954.38
   391.5 1956.18   402.5 1956.26   420.2 1960.43   437.4 1966.87   453.9 1973.94
#Mann= 5 ,-1 , 0
       0      .1       0  121.38     .04       0   174.6    .045       0
   196.6     .04       0  264.66      .1       0
#XS Ineff= 3 ,-1
       0   170.6    1945   200.6     212  1942.5     212   453.9    1945
Permanent Ineff=
       F       F       F
Bank Sta=174.6,196.6
XS Rating Curve= 0 ,0
Exp/Cntr(USF)=0,0
Exp/Cntr=0.5,0.3

Type RM Length L Ch R = 1 ,5162    ,334,342.5,347.1
XS GIS Cut Line= 3
2021955.51411276270330.0908774462022153.13034699  270233.5542113
2022335.98214993269997.323310612
#Sta/Elev= 30
       0 2021.46     7.3 2018.14    14.6 2015.73    32.9 2011.31   119.5 1985.98
   138.8 1979.78   146.1 1977.06     179 1961.68   193.1 1956.63   229.4 1947.53
   262.2 1942.47     267 1940.07   278.5 1932.71   293.8 1928.63   299.6 1928.02
   311.3 1928.89   318.3 1930.85   324.8 1931.45   339.3 1934.51   355.7  1933.6
   360.4 1934.43   366.3 1935.89   378.7 1936.59   384.9 1937.84   411.8 1947.88
   460.9 1954.58     476 1957.11   486.7 1960.74   499.1 1965.58   518.7 1975.75
#Mann= 5 ,-1 , 0
       0      .1       0   293.8    .045       0   311.3      .1       0
   360.4     .04       0   460.9      .1       0
Bank Sta=293.8,311.3
XS Rating Curve= 0 ,0
Exp/Cntr(USF)=0,0
Exp/Cntr=0.3,0.1

Type RM Length L Ch R = 1 ,4819    ,280.3,262.3,248.1
XS GIS Cut Line= 2
2022060.98394066270554.4682551532022616.93223392270300.788197064
#Sta/Elev= 30
       0 2032.08    28.4 2016.29   111.3 1974.48   125.7 1965.95   143.5 1958.44
   165.8 1951.22   185.6 1946.34   197.4 1944.56   227.7 1942.08   266.4 1936.74
   273.6 1933.82   280.8  1929.8   293.2 1918.26   295.2 1917.07   298.8 1916.56
   316.9 1918.41   324.1 1920.54   334.9  1920.9   341.6 1922.11   349.3 1927.18
   352.9 1928.57   367.3 1928.94     407 1942.48   439.5 1947.16   464.7 1949.56
   518.8 1962.58   530.3 1964.29   540.4 1967.77   557.1 1971.77   611.1 1987.61
#Mann= 4 ,-1 , 0
       0      .1       0   293.2    .045       0   316.9     .04       0
     410      .1       0
#XS Ineff= 2 , 0
                             327            1924
Permanent Ineff=
       F       F
Bank Sta=293.2,316.9
XS Rating Curve= 0 ,0
Exp/Cntr=0.3,0.1

Type RM Length L Ch R = 1 ,4557    ,192.3,197.2,200.4
XS GIS Cut Line= 4
2022212.12817645270848.3383538412022349.61085574270770.752365268
2022478.58252904270544.7523732042022671.80825546270430.704391943
#Sta/Elev= 30
       0 2002.51    22.8 1991.18    36.9 1983.28    49.3 1977.75    74.6 1964.29
   142.4 1936.67   157.4 1925.64   169.3 1918.28   176.8 1914.74   186.5 1912.74
   243.2 1914.33   251.4 1914.13   256.4 1912.74   265.9 1911.97   286.4 1912.32
   293.9 1913.36   301.5 1917.03   305.2 1917.92   335.5  1919.7   347.6 1923.01
   361.9 1924.07   371.7  1923.8   386.1 1925.89   435.5 1928.74   464.1 1932.31
   482.1 1935.74   520.4 1947.57   546.7 1957.86   606.6 1978.29   642.4 1992.95
#Mann= 3 ,-1 , 0
       0      .1       0   256.4    .045       0   293.9      .1       0
#XS Ineff= 2 , 0
             243    1918
Permanent Ineff=
       F       F
Bank Sta=256.4,293.9
XS Rating Curve= 0 ,0
Exp/Cntr=0.3,0.1

Type RM Length L Ch R = 1 ,4360    ,246.3,246.7,243.8
XS GIS Cut Line= 3
2022345.99721518270963.9839612742022651.62498001270695.233196439
 2022708.5979619270580.509019363
#Sta/Elev= 30
       0 1976.96    25.3 1963.25    60.2 1948.52    83.5 1940.16     109 1929.05
   128.7 1922.21   152.9  1915.9   164.8 1910.17   183.4 1907.44   218.4 1903.43
   238.1 1902.16   248.5 1900.53   253.2 1901.03   267.1 1906.09   272.8 1906.79
   292.7 1906.28   299.7 1902.17     309 1900.75   315.9 1902.53   322.5 1906.05
   341.5 1906.16   349.5 1909.47   371.7 1914.12   385.7 1917.99     409  1922.4
     429  1927.9   444.6 1933.69   479.5 1950.05   516.7 1966.03   535.1 1971.69
#Mann= 5 ,-1 , 0
       0      .1       0   299.7    .045       0   315.9      .1       0
     350     .04       0  476.98      .1       0
#XS Ineff= 2 , 0
             280    1908     330            1908
Permanent Ineff=
       F       F
Bank Sta=299.7,315.9
XS Rating Curve= 0 ,0
Exp/Cntr=0.3,0.1

Type RM Length L Ch R = 1 ,4113    ,288.5,297.8,310.6
XS GIS Cut Line= 4
2022380.85794145271097.8116614672022628.24123627271032.690170525
2022782.36542274270886.2363396662022936.29215788270805.841307627
#Sta/Elev= 30
       0 1988.27       8 1985.63      25 1976.69    45.3  1969.3    65.7 1960.57
     103 1939.78   123.4 1931.14   150.5 1922.41   194.6 1912.83   231.9 1908.03
   269.3 1906.33   290.2 1902.64   309.9 1897.33     319 1896.46     332 1896.87
   352.9  1892.4   362.1 1890.68   373.3  1891.2   377.8 1892.35   383.7    1895
   392.3 1895.86   400.5 1898.05   418.6 1899.43   427.1 1904.11   479.5 1923.49
   520.2 1944.32   549.8  1957.6   617.2 1994.72   634.2 2003.14   642.1  2006.1
#Mann= 5 ,-1 , 0
       0      .1       0   352.9    .045       0   377.8      .1       0
  395.81     .04       0  528.42      .1       0
Bank Sta=352.9,377.8
XS Rating Curve= 0 ,0
Exp/Cntr=0.3,0.1

Type RM Length L Ch R = 1 ,3815    ,213.4,207.9,203.1
XS GIS Cut Line= 3
2022457.56177912271275.9207463712022874.00701128  271224.4919015
2023056.96181884271165.516937732
#Sta/Elev= 30
       0 1962.03     9.9 1957.24    26.4 1951.94    66.1 1933.32    82.9 1927.21
   128.9 1917.53   148.7  1914.6   171.8 1907.82     195 1899.59   218.1 1893.98
   247.9 1891.24   254.5 1889.16   261.1 1885.34   264.4 1883.81   267.7 1883.44
   277.6 1883.63   286.6 1885.02   308.9 1886.82   340.4 1886.99   363.6 1893.69
   380.1 1896.51   393.3 1899.51   436.2 1914.25   446.6  1918.6   487.2 1933.26
   522.2 1946.84   554.2 1957.49   578.4 1968.39     603 1980.73   611.8  1984.4
#Mann= 3 ,-1 , 0
       0      .1       0   261.1    .045       0   286.6      .1       0
#XS Ineff= 2 , 0
                             312            1892
Permanent Ineff=
       F       F
Bank Sta=261.1,286.6
XS Rating Curve= 0 ,0
Exp/Cntr=0.3,0.1

Type RM Length L Ch R = 1 ,3607    ,244.3,255.8,262.7
XS GIS Cut Line= 2
2022555.32400504271546.145682388 2023073.9719761271315.214833959
#Sta/Elev= 30
       0 1949.58    46.1 1929.57    68.9 1921.58    78.4 1917.05   122.8 1908.21
   133.6 1904.26   197.7 1889.03   212.6 1887.38     220  1883.3   226.9 1880.94
   254.8 1878.71   266.4 1877.06   277.1  1878.3   284.4  1882.2   287.1 1882.57
   309.4 1880.57   320.3 1881.08   327.5 1880.41   359.8 1886.88   384.9 1887.78
   401.4 1895.21   413.7 1901.96   448.6 1925.31   471.1 1937.88   484.4 1943.18
   496.3 1946.15   517.8 1950.12   532.2 1951.14   551.4 1960.37   567.7  1971.8
#Mann= 5 ,-1 , 0
       0      .1       0   254.8    .045       0   277.1      .1       0
     300     .04       0     410      .1       0
#XS Ineff= 2 , 0
             233    1885     295            1885
Permanent Ineff=
       F       F
Bank Sta=254.8,277.1
XS Rating Curve= 0 ,0
Exp/Cntr(USF)=0,0
Exp/Cntr=0.3,0.1

Type RM Length L Ch R = 1 ,3351    ,186.7,194.9,200.5
XS GIS Cut Line= 3
2022575.51468031 271647.099058752023041.16212879271649.622893159
2023177.44918688271573.907860888
#Sta/Elev= 30
       0 1956.16     6.7 1952.75    29.1 1944.27    40.1 1936.94      46 1933.98
    59.2 1930.46    75.6 1924.02   108.4 1913.34   137.9 1898.44     174  1888.8
   210.1 1881.89   242.9 1879.05   318.4 1875.77     337 1871.18   351.2 1869.13
     361 1869.43   366.7 1871.23   377.4 1877.07   390.5  1878.3   397.1 1878.02
   406.9 1883.64   429.9 1890.52   452.9  1899.9   489.8 1913.22   506.7 1918.25
   534.9 1928.45   544.9 1930.95   574.2 1941.39   586.6 1944.58   621.6 1955.81
#Mann= 4 ,-1 , 0
       0      .1       0     337    .045       0   366.7     .04       0
     450      .1       0
Bank Sta=337,366.7
XS Rating Curve= 0 ,0
Exp/Cntr(USF)=0,0
Exp/Cntr=0.3,0.1

Type RM Length L Ch R = 1 ,3157    ,177,180.3,182.5
XS GIS Cut Line= 4
2022538.03737636271720.388503227 2022713.2608333 271734.46812041
2023062.61472126271919.673174929 2023242.3447387271863.504355888
#Sta/Elev= 30
       0 1986.45    47.6 1958.62      70 1946.47    97.5 1933.42   106.8 1927.21
     120 1923.35   139.7 1913.18   179.7 1896.27     202 1890.13   235.4 1879.05
   256.6 1874.51   276.2 1872.63   303.6 1870.41   317.2 1870.56   343.9 1868.02
   385.2 1867.41   392.5 1866.11   404.6 1864.95   409.5  1866.2   416.7 1869.95
     421 1870.56   438.6  1870.7     447 1872.16   506.5 1876.73   564.8 1885.61
   645.3 1900.71   691.1 1912.54     698 1915.37   734.7 1934.29   759.5 1942.94
#Mann= 5 ,-1 , 0
       0      .1       0  365.79     .04       0   392.5    .045       0
   409.5     .04       0  535.79      .1       0
#XS Ineff= 2 , 0
             368    1872
Permanent Ineff=
       F       F
Bank Sta=392.5,409.5
XS Rating Curve= 0 ,0
Exp/Cntr=0.3,0.1

Type RM Length L Ch R = 1 ,2976    ,232.9,224.5,214.6
XS GIS Cut Line= 4
2022544.69430648 271878.925134432022708.59931182271899.513719342
2022940.20875242272088.7700803362023168.22824839 272086.37829891
#Sta/Elev= 30
       0 1998.43     4.7 1997.21    17.9 1986.43    60.9 1955.69    70.8 1950.69
    80.8 1946.87    87.1 1943.13   127.1 1913.13   143.6  1902.1   156.8  1892.2
   173.1 1883.21   188.4 1873.38   196.8 1868.71   203.4  1866.3   237.5 1860.62
   245.4 1857.78   247.8 1856.99   258.2 1856.52   261.7 1857.15   268.7 1860.66
   273.1 1861.96   294.3 1865.03   311.2 1863.88     320    1866   374.8 1864.22
   421.4 1869.26   480.3 1872.83   503.3 1875.65   617.2 1893.25   692.3 1903.17
#Mann= 5 ,-1 , 0
       0      .1       0   245.4    .045       0   261.7      .1       0
  325.19     .04       0  455.19      .1       0
Bank Sta=245.4,261.7
XS Rating Curve= 0 ,0
Exp/Cntr=0.3,0.1

Type RM Length L Ch R = 1 ,2752    ,220.9,226.7,231.2
XS GIS Cut Line= 3
2022543.42341287272097.5369741832022667.63463625 272159.43744379
2023141.95940752272154.529305364
#Sta/Elev= 30
       0 2004.72      14  1995.9    21.3 1990.38      36 1982.29    83.6 1946.83
   131.3 1905.15   150.9  1886.4   164.9 1874.97   174.7 1868.54   187.8 1861.61
   197.3 1855.22   207.8 1853.68   220.7 1851.53   223.9 1851.56   227.2 1852.64
   227.2 1852.66   233.7 1854.71   250.2 1857.36   273.2 1857.41   286.3 1860.43
   299.4 1859.65   319.1 1860.39   358.5 1862.76   401.1 1867.59   437.2 1868.46
     447 1871.01   467.6 1873.42   506.5 1883.24   535.8  1887.1   613.1 1899.42
#Mann= 4 ,-1 , 0
       0      .1       0   207.8    .045       0   227.2     .04       0
  398.78      .1       0
Bank Sta=207.8,227.2
XS Rating Curve= 0 ,0
Exp/Cntr=0.3,0.1

Type RM Length L Ch R = 1 ,2525    ,181.9,177.7,172.2
XS GIS Cut Line= 3
2022475.76856132272183.6538913872022556.58592225 272320.96284597
 2022976.3071075272469.418904296
#Sta/Elev= 30
       0 2004.59    47.4 1982.71    73.6 1967.39   107.8 1941.84   119.3 1935.16
   162.1 1899.26   186.5 1882.33   208.9 1864.77   216.6 1860.01     232 1853.19
   238.7 1851.91   290.9 1849.72   311.7    1850     322 1847.24   329.2 1846.09
   341.1 1847.18     350 1849.44   367.4 1850.35     394 1855.69   409.2 1855.48
   419.7 1856.85     451 1855.92     484 1857.74   494.2  1854.7   513.6 1859.53
   527.7 1859.51     531  1860.3   555.4 1872.95   593.6 1885.93   604.5 1887.48
#Mann= 6 ,-1 , 0
       0      .1       0     322    .045       0   341.1      .1       0
  349.33     .04       0  429.33      .1       0  559.33     .04       0
#XS Ineff= 2 , 0
             300    1855
Permanent Ineff=
       F       F
Bank Sta=322,341.1
XS Rating Curve= 0 ,0
Exp/Cntr=0.3,0.1

Type RM Length L Ch R = 1 ,2347    ,179.7,191.3,203.5
XS GIS Cut Line= 3
2022442.80230006272435.3730056392022567.97319675272548.600917205
2022907.39890511272558.203280421
#Sta/Elev= 30
       0 1884.26      42 1869.73      56 1867.23    64.1 1865.02    97.8 1859.42
   139.3 1854.08   186.3 1849.82   199.4 1846.92   225.7 1846.99   245.4 1843.09
   271.6 1844.06     285 1841.66   297.9 1840.59   311.5  1841.8   317.6 1842.69
     334  1847.2   343.8 1847.74     357 1847.41   363.5 1849.39   396.8 1847.73
     400 1848.42   422.6 1859.03     439 1865.11   445.6  1866.5     462 1867.24
   471.8  1868.5     485 1871.65   494.8 1877.55   498.1 1878.74   508.3 1879.84
#Mann= 4 ,-1 , 0
       0      .1       0     285    .045       0   311.5      .1       0
  338.78     .04       0
#XS Ineff= 2 , 0
             270    1846
Permanent Ineff=
       F       F
Bank Sta=285,311.5
XS Rating Curve= 0 ,0
Exp/Cntr=0.3,0.1

Type RM Length L Ch R = 1 ,2156    ,208.7,214.3,216.3
XS GIS Cut Line= 2
2022339.51030462272477.1803612482022774.24185159272852.885918417
#Sta/Elev= 30
       0 1897.42    17.2 1887.16    29.8 1881.26    62.4 1867.82   113.6  1854.1
   129.9 1852.18     169  1849.7   230.1  1847.4   276.4 1844.31   295.3  1842.1
     309 1841.61   320.7 1838.53   330.5 1837.18   355.4  1838.5   372.8 1837.64
   380.6 1836.97   390.7 1837.08   395.7 1837.85   403.1 1840.23   425.8 1841.54
   436.9 1840.57   439.2 1841.38   446.2 1847.06   453.2 1850.02   457.8 1852.98
   476.4 1871.44   490.4 1882.37   506.1 1892.89   536.9 1909.82   574.6 1927.53
#Mann= 4 ,-1 , 0
       0      .1       0   372.8    .045       0   395.7     .04       0
     520      .1       0
Bank Sta=372.8,395.7
XS Rating Curve= 0 ,0
Exp/Cntr=0.3,0.1

Type RM Length L Ch R = 1 ,1942    ,160.8,168.3,172.2
XS GIS Cut Line= 3
2022277.91571686272542.1449852432022347.60548001272682.337735113
 2022610.7710204273006.762813197
#Sta/Elev= 30
       0 1892.82    18.5 1883.14    29.5 1879.02    50.9  1872.7    60.7 1871.58
    72.9 1868.03   170.6  1849.9   237.8 1841.78   259.3 1836.85   267.8 1835.96
   289.4 1835.78   297.4 1834.06   307.8 1829.82   317.1 1828.88   326.4  1829.4
   328.8 1830.31   331.2 1831.33   343.8 1832.99   352.3 1836.31   360.7  1837.4
   391.7 1836.95   424.1 1835.18   436.8 1839.36   453.7 1852.73   466.4 1864.45
   470.6 1868.89   474.8 1874.52     478 1877.19   521.3 1903.09   574.3 1939.28
#Mann= 5 ,-1 , 0
       0      .1       0   307.8    .045       0   328.8     .06       0
  446.56     .04       0  456.56      .1       0
Bank Sta=307.8,328.8
XS Rating Curve= 0 ,0
Exp/Cntr=0.3,0.1

Type RM Length L Ch R = 1 ,1773    ,345.4,325.1,299.9
XS GIS Cut Line= 4
2022143.06316989272644.1410837432022242.53940191272706.182518797
2022352.46799544273044.6314291542022444.72030354273111.325829034
#Sta/Elev= 30
       0  1914.1    12.2 1904.48    30.3 1891.78    76.7 1865.83   105.2 1857.38
   141.6 1850.27     183 1838.01     214 1832.73   238.2 1830.73   255.4 1830.33
   276.1 1825.73     283 1824.85   286.5  1824.9   290.6 1826.02   295.8  1828.3
     301 1829.62   331.3 1832.05   365.8 1832.62   372.7 1831.06   386.5 1830.39
     390 1828.95   393.4  1830.8   400.3 1836.48   433.8 1844.96   462.5 1854.31
   465.9 1855.99   473.1 1860.97   497.5  1871.7   539.7 1891.92   586.9 1911.69
#Mann= 6 ,-1 , 0
       0      .1       0   276.1    .045       0   290.6      .1       0
  327.24     .06       0  427.24     .04       0  437.24      .1       0
#XS Ineff= 2 , 0
             245    1836     305            1836
Permanent Ineff=
       F       F
Bank Sta=276.1,290.6
XS Rating Curve= 0 ,0
Exp/Cntr=0.3,0.1

Type RM Length L Ch R = 1 ,1448    ,320,336.6,350.6
XS GIS Cut Line= 4
2021900.51578595272990.0844745262021975.03073496273034.048294442
2022267.87448457273042.9900883232022370.70511421273135.388625096
#Sta/Elev= 30
       0 1892.22    14.4  1882.7      22 1876.68    53.4 1855.52    86.5 1836.57
    99.9 1833.75   109.4 1833.09   120.1 1834.12   145.8 1834.75   172.1 1832.74
   175.3 1831.96   198.3 1821.78   211.4 1819.81     218  1818.5   224.6 1818.27
   234.4 1818.73   244.3 1820.37   254.1 1823.53   257.4 1823.87   283.7 1823.53
   303.7 1824.68   338.7 1824.48   349.3 1829.61   391.3 1836.97   421.8 1851.76
   425.7 1853.89   435.7 1861.28     445 1866.07   477.5 1881.57   517.7 1899.01
#Mann= 5 ,-1 , 0
       0      .1       0   211.4    .045       0   244.3      .1       0
  256.52     .06       0  356.52      .1       0
Bank Sta=211.4,244.3
XS Rating Curve= 0 ,0
Exp/Cntr(USF)=0,0
Exp/Cntr=0.3,0.1

Type RM Length L Ch R = 1 ,1112    ,262.3,258.9,252.9
XS GIS Cut Line= 2
2021740.30864558273078.7572638482022164.29870545273359.678621617
#Sta/Elev= 30
       0 1901.73    33.9 1885.94    73.2 1861.94   111.5 1843.83   115.8 1840.18
   121.8 1831.67   124.4 1828.65   132.3 1822.99   142.3  1814.7     147 1811.93
   156.5 1810.37     166 1810.97   170.7 1812.11   177.8 1813.34   193.1 1812.63
   203.1 1813.36   215.7 1812.92   240.6 1814.77   270.1 1814.39     294 1817.37
   321.2 1817.43   356.6 1819.75   383.1 1819.83   402.7 1827.21   419.6 1835.15
   439.2 1845.72     451 1855.17     469 1862.98   485.5  1872.2   508.6 1882.85
#Mann= 5 ,-1 , 0
       0      .1       0     147    .045       0   170.7      .1       0
     360     .04       0     400      .1       0
#XS Ineff= 2 , 0
                             227            1818
Permanent Ineff=
       F       F
Bank Sta=147,170.7
XS Rating Curve= 0 ,0
Exp/Cntr(USF)=0,0
Exp/Cntr=0.3,0.1

Type RM Length L Ch R = 1 ,853     ,263.7,261.7,258.3
XS GIS Cut Line= 2
2021581.59180419273320.1856986422022112.88339063273513.924566069
#Sta/Elev= 30
       0 1894.72    20.9  1880.9    34.9 1874.63      56 1862.18    97.7  1841.2
   102.1  1837.7   104.7 1833.94   111.7 1819.22   115.2 1816.05   127.7  1811.4
   148.2 1806.37   157.1 1804.97     171 1805.02     178 1806.47   188.5 1807.31
     199 1812.74   209.5 1814.09   233.9 1813.08   345.7 1814.32   373.6 1816.06
   386.1 1821.08     405 1821.17   409.2 1823.08   422.5 1832.75   443.4  1841.7
     468  1855.1   499.3 1868.64   521.8 1877.27   537.7 1881.98   565.5 1887.01
#Mann= 5 ,-1 , 0
       0      .1       0   148.2    .045       0     178      .1       0
     390     .06       0     490      .1       0
Bank Sta=148.2,178
XS Rating Curve= 0 ,0
Exp/Cntr(USF)=0,0
Exp/Cntr=0.3,0.1

Type RM Length L Ch R = 1 ,591     ,62.9,63.8,63.8
XS GIS Cut Line= 2
2021524.96044294 273596.636159472021922.87027065 273667.42536103
#Sta/Elev= 30
       0 1859.85    24.1 1848.53    44.1 1837.17    57.5 1830.63    64.8  1826.5
    74.1 1820.02    90.8 1811.27   107.4 1804.96   114.1 1801.34   117.4 1800.18
   127.4 1798.82   137.4  1797.2     144 1797.46   147.4 1798.18   154.1 1801.07
   160.8 1802.92   194.1 1804.09   230.7 1808.21   268.5 1810.51   327.4 1815.88
     334  1814.7   350.5 1814.63   357.4 1819.65   367.2 1825.25   380.7 1830.98
     384 1833.01   390.7  1840.8     394 1843.52   399.6 1845.79   404.2 1846.94
#Mann= 4 ,-1 , 0
       0      .1       0   127.4    .045       0   147.4      .1       0
     330     .04       0
#XS Ineff= 2 , 0
                             175            1810
Permanent Ineff=
       F       F
Bank Sta=127.4,147.4
XS Rating Curve= 0 ,0
Exp/Cntr(USF)=0,0
Exp/Cntr=0.5,0.3

Type RM Length L Ch R = 1 ,527     ,20.7,20.6,20.8
XS GIS Cut Line= 2
2021563.85255236273664.1864487462021854.01103171273726.225108793
#Sta/Elev= 30
       0 1824.49    16.7 1814.69    31.5 1808.38    34.9    1806    38.2 1804.18
    51.6 1802.22    62.1 1801.64    71.8 1802.12    75.1 1801.91    78.5 1801.06
    84.2 1797.82    88.5 1796.43    98.6  1796.3     102 1797.16   102.91797.749
   108.7 1801.49     112 1802.55   118.7 1802.18   131.2 1800.62   162.3 1801.58
   182.5 1804.08     192 1804.67   229.4 1806.89   242.9 1808.35   259.6 1810.69
   269.7 1811.08   279.8 1810.73   283.2 1811.42   288.7 1814.37   296.7 1817.81
#Mann= 5 ,-1 , 0
       0      .1       0    84.2    .045       0   102.9      .1       0
   131.2    .035       0     192     .04       0
#XS Ineff= 3 ,-1
       0    76.2  1802.9   110.9     115  1800.5     115  296.72  1802.9
Permanent Ineff=
       F       F       F
Bank Sta=84.2,102.9
XS Rating Curve= 0 ,0
Exp/Cntr(USF)=0,0
Exp/Cntr=0.5,0.3

Type RM Length L Ch R = 1 ,507     ,121.2,121.1,121
XS GIS Cut Line= 2
2021545.69419164273682.0561232772021853.63573967273745.855769021
#Sta/Elev= 30
       0 1830.49     6.4 1825.81    16.5 1819.51    19.8 1817.83    26.5 1815.42
    37.6 1810.77    46.6    1806    48.7 1805.21    53.3 1804.64    66.8 1804.55
    80.2 1802.57    86.9 1801.11    96.9 1796.62   100.3 1795.95   113.7 1795.71
     117 1795.77   120.4 1796.38   123.7 1798.34   127.1 1799.71   170.6 1800.66
     184 1801.43   201.3  1803.3   210.8 1803.83   247.7 1806.84   264.4  1809.9
   277.8 1810.43   287.9 1809.85   291.2 1810.49   297.9 1813.62   314.5 1820.35
#Mann= 4 ,-1 , 0
       0      .1       0    96.9    .045       0   120.4    .035       0
   210.8     .04       0
#XS Ineff= 3 ,-1
       0    91.9    1802   126.4     135  1799.3     135 334.595    1802
Permanent Ineff=
       F       F       F
Bank Sta=96.9,120.4
XS Rating Curve= 0 ,0
Exp/Cntr(USF)=0,0
Exp/Cntr=0.5,0.3

Type RM Length L Ch R = 1 ,386     ,163.9,174.8,186.9
XS GIS Cut Line= 2
2021487.50405875 273794.019834252021819.10128099273860.860112011
#Sta/Elev= 30
       0 1834.08     8.8 1833.16    12.2 1832.32    35.7  1822.1      39 1819.16
    42.4 1814.42    45.7  1810.5    49.1 1808.97    95.1 1801.29   107.7 1799.88
   129.4 1798.37   136.9  1794.7   139.4 1794.15   146.1    1794   156.2  1794.2
   159.2 1794.74   166.2 1796.31   172.9 1796.94     193 1798.08   216.4 1797.81
   236.5 1800.85   259.9 1802.98   281.7 1804.14   293.4 1803.84   295.7 1804.24
   300.1 1806.43   306.8 1811.11   323.6 1819.02   333.5 1824.87   338.3 1826.68
#Mann= 4 ,-1 , 0
       0      .1       0   136.9    .045       0   159.2      .1       0
     170     .04       0
#XS Ineff= 2 , 0
                          196.89         1801.84
Permanent Ineff=
       F       F
Bank Sta=136.9,159.2
XS Rating Curve= 0 ,0
Exp/Cntr(USF)=0,0
Exp/Cntr=0.3,0.1

Type RM Length L Ch R = 1 ,211     ,55.1,56,57.5
XS GIS Cut Line= 3
2021438.02489206 273817.457334252021535.24711433273945.929556459
 2021783.5110032273939.853167579
#Sta/Elev= 30
       0 1847.62     9.6 1845.63    18.9 1842.07    30.2 1841.93      33 1841.21
    47.5 1833.74    58.8 1828.67    65.8  1824.7    75.5 1820.31    79.6 1817.87
    84.5 1813.31    96.1 1804.44   100.2 1797.52   103.2 1791.31   105.6 1788.87
   108.4 1787.77     115 1787.11   120.7  1787.3   126.7 1788.66   145.4 1793.57
   157.1 1794.29     168 1795.95   236.9 1796.06   286.2 1796.85   325.6 1799.35
   361.7 1800.57   374.8 1800.19   378.1 1800.95   387.9 1806.85   409.5 1815.82
#Mann= 4 ,-1 , 0
       0      .1       0   105.6    .045       0   126.7      .1       0
  371.11     .04       0
Bank Sta=105.6,126.7
XS Rating Curve= 0 ,0
Exp/Cntr(USF)=0,0
Exp/Cntr=0.3,0.1

Type RM Length L Ch R = 1 ,155     ,129.7,154.8,163.2
XS GIS Cut Line= 3
2021421.70786992273887.5203465752021530.53973408274023.182543456
 2021432.4192868274357.093841403
#Sta/Elev= 30
       0 1844.62       9 1842.88    27.3 1833.33      42 1823.25      53 1810.32
    56.2 1805.25    62.3 1792.24    67.3 1787.16    71.9 1785.82    83.3 1784.88
    99.7 1786.65   104.3 1789.03   109.3 1789.89   120.7 1786.26     143 1786.19
   155.6  1789.4   168.2  1790.3   227.4 1789.77   251.3 1791.53   295.8 1791.15
   360.8 1792.33   439.4 1795.85   455.7 1798.51   466.8 1804.16   483.9 1804.94
   487.3 1806.15   497.5 1816.87     501 1819.95   504.4 1821.52     522 1821.29
#Mann= 4 ,-1 , 0
       0      .1       0    67.3    .045       0    99.7      .1       0
  343.92     .04       0
#XS Ineff= 2 , 0
                          108.51            1792
Permanent Ineff=
       F       F
Bank Sta=67.3,99.7
XS Rating Curve= 0 ,0
Exp/Cntr(USF)=0,0
Exp/Cntr=0.3,0.1

Type RM Length L Ch R = 1 ,0       ,,,
XS GIS Cut Line= 2
2021375.17812102273906.1103895062021333.14589584274358.440150179
#Sta/Elev= 30
       0 1846.98      11 1844.84    20.8 1841.63    27.4 1841.41    30.7 1840.73
    37.3 1836.56    47.2 1832.43    50.5 1830.54    73.6 1815.06    93.3 1804.32
    96.6 1802.08    99.9 1798.95   103.2 1794.69   106.5 1788.58   109.8  1783.5
   113.1  1781.7   136.2    1780   142.8 1781.49   152.6 1784.49   162.5 1785.47
   188.9  1787.2   254.8 1788.95   277.8 1790.04   343.7 1795.99     380 1798.65
   403.1 1800.06   409.6 1801.28   416.2  1805.4     436 1806.91   454.3 1809.52
#Mann= 4 ,-1 , 0
       0      .1       0   113.1    .045       0   142.8      .1       0
     380     .06       0
#XS Ineff= 2 , 0
                             159          1787.5
Permanent Ineff=
       F       F
Bank Sta=113.1,142.8
XS Rating Curve= 0 ,0
Exp/Cntr(USF)=0,0
Exp/Cntr=0.3,0.1
LCMann Table=0

Chan Stop Cuts=-1
Use User Specified Reach Order=0
Composite Channel Slope=5
